--- FudgesCr.prj (project) ---

Proj Title=FudgesCr
Current Plan=p01
Geom File=g01
Flow File=f01
Plan File=p01
DSS Export Rating Curves=0
DSS Export Rating Curve Sorted=0
DSS Export Volume Flow Curves=0
DXF OffsetX=0
DXF OffsetY=0
DXF ScaleX=0
DXF ScaleY=0

--- FudgesCr.p01 (plan) ---

Plan Title=Floodplain
Program Version=4.00
Geom File=g01
Flow File=f01
K Sum by GR=0
Std Step Tol=0.01
Critical Tol=0.01
Num of Std Step Trials=20
Max Error Tol=0.3
Flow Tol Ratio=0.001
Split Flow NTrial=30
Split Flow Tol=0.02
Split Flow Ratio=0.02
Log Output Level=0
Friction Slope Method=1
Unsteady Friction Slope Method=2
Unsteady Bridges Friction Slope Method=1
Global Log Level=0
CheckData=False
Run HTab=0
Run UNet=0
Run PostProcess=0
UNET Theta=0
UNET Theta Warmup=0
UNET ZTol=0
UNET ZSATol=0
UNET MxIter=0
UNET MaxInSteps=0
UNET DtIC=0
UNET DtMin=0
UNET MaxCRTS=0
UNET WFStab=0
UNET SFStab=0
UNET WFX=0
UNET SFX=0
UNET DSS MLevel=0
UNET DZMax Abort=0
UNET Convert EG Bridges=0
UNET Use Existing IB Tables=0
UNET Froude Limit=0
UNET Froude Power=0
Write IC File=0
Echo Input=False
Echo Output=False
Write Detailed=0

--- FudgesCr.f01 (steady flow) ---

Flow Title=NFF Regression Equation
Program Version=4.10
Number of Profiles= 1
Profile Names=P100yr
River Rch & RM=FudgesCr,Main            ,25028.3
     887
River Rch & RM=FudgesCr,Main            ,24670.4
     890
River Rch & RM=FudgesCr,Main            ,24180.9
     906
River Rch & RM=FudgesCr,Main            ,23267.7
     933
River Rch & RM=FudgesCr,Main            ,22877.7
     944
River Rch & RM=FudgesCr,Main            ,21729.3
     954
River Rch & RM=FudgesCr,Main            ,21303.2
    1082
River Rch & RM=FudgesCr,Main            ,20973
    1089
River Rch & RM=FudgesCr,Main            ,20656.4
    1193
River Rch & RM=FudgesCr,Main            ,19357
    1206
River Rch & RM=FudgesCr,Main            ,18416.7
    1234
River Rch & RM=FudgesCr,Main            ,17913.8
    1338
River Rch & RM=FudgesCr,Main            ,17151
    1346
River Rch & RM=FudgesCr,Main            ,16508.5
    1440
River Rch & RM=FudgesCr,Main            ,16039.8
    1485
River Rch & RM=FudgesCr,Main            ,15469.9
    1509
River Rch & RM=FudgesCr,Main            ,15304.1
    1527
River Rch & RM=FudgesCr,Main            ,13747.9
    1558
River Rch & RM=FudgesCr,Main            ,13171
    1614
River Rch & RM=FudgesCr,Main            ,12458.4
    1619
River Rch & RM=FudgesCr,Main            ,12203.4
    2068
River Rch & RM=FudgesCr,Main            ,10806.5
    2125
River Rch & RM=FudgesCr,Main            ,9755.8
    2136
River Rch & RM=FudgesCr,Main            ,8934.5
    2142
River Rch & RM=FudgesCr,Main            ,7704.4
    2179
River Rch & RM=FudgesCr,Main            ,6965.8
    2187
River Rch & RM=FudgesCr,Main            ,6579.8
    2192
Boundary for River Rch & Prof#=FudgesCr,Main            , 1
Up Type= 0
Dn Type= 3
Dn Slope=0.00123
DSS Import GetInterval= 0
DSS Import GetPeak= 0
DSS Import FillOption= 0

--- FudgesCr.g01 (geometry) ---

Geom Title=USGS 10m DEM
Program Version=4.10

River Reach=FudgesCr        ,Main
Reach XY= 30
     1630676.056      510606.185     1630106.255      510527.755
       1629028.7      510708.204     1627801.642      510341.652
     1627525.234      510401.618     1627183.503      510963.325
     1626680.279      511087.302     1626494.324      510983.365
     1625894.416      511307.867      1625010.59      511418.707
     1624717.319       511846.58     1624444.889      511785.462
     1624063.922      511957.114     1622575.862      514277.757
     1622079.903      514717.147      1621705.88      515721.615
     1621822.558      515889.372      1621735.01      516356.123
     1622028.526      516534.819     1622117.824      517369.896
     1622671.187      517913.142     1623087.675      519149.476
     1623036.638      519440.052     1624362.022      520816.033
     1624693.832       521483.38       1623568.8      522513.457
     1622930.579       523496.15     1622434.428       523657.92
     1622271.614       524603.16     1621744.169      524948.786

Type RM Length L Ch R = 1 ,25028.3 ,359.6,357.9,355.9
XS GIS Cut Line= 2
     1630655.439      510494.939     1630643.287        510762.3
#Sta/Elev= 18
       0  687.34    19.1  677.33    28.7  672.51    38.2  668.02    47.8  664.09
    66.9  656.97      86  650.16    95.6  646.91   103.9  645.13   105.1  644.87
   114.7  644.54   118.9  644.84   124.3  645.22   133.8  646.11   143.4  646.61
   219.8  649.63   229.4  650.17   267.6  652.74
#Mann= 3 , 0 , 0
       0      .1       0   103.9    .045       0   118.9     .06       0
Bank Sta=103.9,118.9
XS Rating Curve= 0 ,0
Exp/Cntr=0.3,0.1

Type RM Length L Ch R = 1 ,24670.4 ,498.2,489.5,479.4
XS GIS Cut Line= 2
     1630304.088      510479.557     1630291.067       510812.89
#Sta/Elev= 21
       0  662.01    19.6  658.76    29.4  656.86    39.2  654.24    58.9  647.65
    68.7  645.26    78.5  643.71    88.3  642.71    98.1  642.04   107.9   641.7
   117.7  642.05   120.3   642.3   127.6  643.02   137.4  643.81   147.2  644.28
   215.8  647.09   225.7  647.59   235.5  648.31     314  655.53   323.8  656.67
   333.6  658.79
#Mann= 3 , 0 , 0
       0      .1       0    98.1    .045       0   120.3     .06       0
Bank Sta=98.1,120.3
XS Rating Curve= 0 ,0
Exp/Cntr=0.3,0.1

Type RM Length L Ch R = 1 ,24180.9 ,202.3,213,223.6
XS GIS Cut Line= 2
     1629804.745      510515.772     1629965.546      510864.973
#Sta/Elev= 24
       0  655.66     9.6  654.35    57.7  649.67    67.3  647.94    76.9  644.41
    86.5  640.72      96  638.98   105.7  639.35     111  640.18   115.3  640.86
   124.9  642.14   134.6  642.39   144.2  642.23   153.8  642.22   192.2  642.76
   221.1  642.63   249.9  642.96   326.8  644.42   336.4  645.11     346  647.11
   355.6  650.43   365.2  654.54   374.8  659.25   384.4  664.22
#Mann= 3 , 0 , 0
       0      .1       0    86.5    .045       0     111     .06       0
Bank Sta=86.5,111
XS Rating Curve= 0 ,0
Exp/Cntr=0.3,0.1

Type RM Length L Ch R = 1 ,23967.9 ,265.8,263.9,261.8
XS GIS Cut Line= 2
     1629648.495      510573.064     1629634.817      510917.057
#Sta/Elev= 27
       0  663.35     9.8  660.13    19.7  658.09    29.5  656.35    39.3  654.49
    49.2   652.4      59  649.22    68.8  644.02    78.7  638.51    79.9  638.19
    88.5   635.9    98.4  636.45   108.2  638.19     118  639.58   127.9  640.23
   167.2  641.51   216.4  643.51   236.1  644.11   245.9  644.28   255.7  644.33
   285.2  644.24   295.1   644.4   304.9  644.76   314.8  645.35   324.6  646.27
   334.4   647.7   344.3   649.8
#Mann= 3 , 0 , 0
       0      .1       0    79.9    .045       0    98.4     .06       0
Bank Sta=79.9,98.4
XS Rating Curve= 0 ,0
Exp/Cntr=0.3,0.1

Type RM Length L Ch R = 1 ,23704   ,427.4,436.3,444.3
XS GIS Cut Line= 2
     1629374.189      510514.036     1629393.287      510902.925
#Sta/Elev= 23
       0  705.55     9.7  702.53    19.5  698.57    29.2  694.05    38.9  689.36
    48.7  684.53    68.1  674.68    87.6  665.05    97.3  660.44   126.5  647.05
     146  637.31   150.8  635.71   155.7  634.08   165.5  633.43   175.2  634.42
   184.9  635.79   194.7  636.72   204.4  637.14   253.1  638.29     292  639.48
     331  640.44   369.9  641.14   389.4   641.1
#Mann= 3 , 0 , 0
       0      .1       0   150.8    .045       0   175.2     .06       0
Bank Sta=150.8,175.2
XS Rating Curve= 0 ,0
Exp/Cntr=0.3,0.1

Type RM Length L Ch R = 1 ,23267.7 ,389.3,390,388.8
XS GIS Cut Line= 2
     1629018.287        510512.3     1628910.859      510859.765
#Sta/Elev= 24
       0  694.72    19.7  684.89    49.2  669.95    78.6  654.24   108.1   639.2
     118  634.88   127.8  632.37   137.6  631.56   157.3  631.12   176.9  629.76
   177.5  629.78   186.8  630.05   192.5  631.02   196.6  631.72   206.4  633.75
   216.2  634.89   226.1  635.22   245.7  635.56   304.7  637.42   324.4  637.88
   334.2  638.19     344  638.65   353.9  639.23   363.7  639.99
#Mann= 3 , 0 , 0
       0      .1       0   177.5    .045       0   192.5     .06       0
Bank Sta=177.5,192.5
XS Rating Curve= 0 ,0
Exp/Cntr=0.3,0.1

Type RM Length L Ch R = 1 ,22877.7 ,354.4,353.2,352.3
XS GIS Cut Line= 2
     1628638.078      510434.175     1628553.009      510718.897
#Sta/Elev= 24
       0  669.19     9.6  664.54    19.2  660.07    28.8  655.78    38.3  651.64
    47.9  647.71    67.1  640.19    76.7  636.68    86.3  633.75    95.9  631.79
   105.4  630.56     115  629.54   124.6  628.38   134.2  627.34   138.6  627.27
   143.8  627.18   153.6  628.41     163  630.44   172.5  631.99   182.1  632.54
   230.1  633.83   258.8  634.71   287.6  635.87   297.2  636.53
#Mann= 3 , 0 , 0
       0      .1       0   138.6    .045       0   153.6     .06       0
Bank Sta=138.6,153.6
XS Rating Curve= 0 ,0
Exp/Cntr=0.3,0.1

Type RM Length L Ch R = 1 ,22524.5 ,46.8,46.7,46.8
XS GIS Cut Line= 3
     1628422.801      510244.939     1628280.439      510385.564
     1628235.301      510566.119
#Sta/Elev= 28
       0  691.23     9.5  685.78    28.6  674.99    38.1  669.81    47.6  664.79
    95.3   640.5   104.8   635.8   114.4  632.18   123.9  630.27   133.4  629.58
   171.5  627.72     181  627.27   200.1  626.53   219.7  626.22   249.1   626.1
   258.9  625.92   278.5   624.3   280.7  624.31   288.3  624.36   295.7  625.22
   298.1   625.5   307.8  627.14   327.4   629.5   337.2  630.94     347   632.7
   356.8  634.75   376.4  639.13   386.2  641.14
#Mann= 3 , 0 , 0
       0     .06       0   280.7    .045       0   295.7      .1       0
Bank Sta=280.7,295.7
XS Rating Curve= 0 ,0
Exp/Cntr=0.3,0.1

Type RM Length L Ch R = 1 ,22477.7 ,95,96,96.6
XS GIS Cut Line= 3
     1628377.662      510232.786     1628235.301      510373.411
     1628190.162      510553.967
#Sta/Elev= 27
       0  677.85     9.5  671.96    19.1  666.11    28.6  660.53    38.1  655.73
    47.6  651.45    85.8  635.19    95.3  632.11   104.8  630.55   114.4  629.78
   133.4  628.42     162   626.6   171.5  626.22     181  626.13   219.7  626.04
   249.1  626.26   258.9  626.06   278.5  624.11   288.3  623.86   297.1  624.54
   298.1  624.62   307.8  625.99   317.6  627.19   327.4  628.61   337.2  630.58
   376.4  639.69   386.2   641.9
#Mann= 3 , 0 , 0
       0     .06       0   278.5    .045       0   297.1      .1       0
Bank Sta=278.5,297.1
XS Rating Curve= 0 ,0
Exp/Cntr=0.3,0.1

Type RM Length L Ch R = 1 ,22381.7 ,661.3,652.4,609.4
XS GIS Cut Line= 2
     1628309.953      509780.529     1628085.338      510560.286
#Sta/Elev= 30
       0  650.22    48.9  655.01    78.2  655.96   107.5  654.49   166.2  652.99
   185.8  652.04   215.1  651.21   224.9  651.04   244.4  651.44     264  651.05
   293.3   649.2   322.6  645.27   342.2  641.49   371.5  634.59   391.1  631.36
   400.8  630.33   420.4  629.63   547.5  627.38   606.2  626.83   664.8  624.86
   674.6  623.83   684.4  623.12   695.9  623.74   703.9   624.7   713.7  626.43
   723.5  628.92   762.6  642.09   782.1  649.41   791.9  653.89   811.5  663.63
#Mann= 3 , 0 , 0
       0     .06       0   674.6    .045       0   695.9      .1       0
Bank Sta=674.6,695.9
XS Rating Curve= 0 ,0
Exp/Cntr=0.3,0.1

Type RM Length L Ch R = 1 ,21729.3 ,444.8,426.1,403.7
XS GIS Cut Line= 4
     1627521.759       510145.98     1627624.189      510328.272
     1627657.176      510534.869     1627717.939      510623.411
#Sta/Elev= 30
       0   713.2     9.5  709.65      19  706.25      38  699.71      57  693.48
    85.5  684.29   104.6  677.93   123.6  671.04   133.1  667.34   142.6   663.5
   152.1  659.52   161.6  655.38   171.1  651.04   180.6  646.39   190.1  640.65
   199.6  634.24   209.1   628.7   218.6  624.91   228.1  623.07   256.6  619.76
   266.2   618.7   275.7  618.37   285.2  619.16   292.4  620.18   294.7   620.5
   304.2  621.45   361.2  625.51   380.3  627.02   418.3  630.28   525.7  640.32
#Mann= 3 , 0 , 0
       0      .1       0   256.6    .045       0   292.4      .1       0
Bank Sta=256.6,292.4
XS Rating Curve= 0 ,0
Exp/Cntr=0.3,0.1

Type RM Length L Ch R = 1 ,21303.2 ,197.3,206.7,216.3
XS GIS Cut Line= 2
     1627301.273      510619.939     1627585.338       510750.39
#Sta/Elev= 21
       0  627.62    39.1  626.11    78.2  624.15   117.2   622.4     127  621.82
   136.8   620.8   146.5  618.87   156.3  616.71   166.1  615.91   175.8  616.16
   185.6  618.17   195.4  621.22   205.1   623.3   214.9  624.86   234.4  627.47
   244.2   628.6     254  629.62   263.8   630.4   273.5  630.92     293  631.67
   312.6  633.13
#Mann= 3 , 0 , 0
       0      .1       0   156.3    .045       0   175.8      .1       0
Bank Sta=156.3,175.8
XS Rating Curve= 0 ,0
Exp/Cntr=0.3,0.1

Type RM Length L Ch R = 1 ,21096.5 ,119.2,123.5,127.6
XS GIS Cut Line= 2
     1627230.092      510736.258     1627410.648      510932.439
#Sta/Elev= 22
       0  621.02      19  620.98    47.6  621.26    66.7   621.2    95.2  620.47
   123.8  619.59   133.3   619.2   142.8  617.98   152.4   616.3   156.9  615.85
   161.9  615.34   171.4   615.8   171.9  615.88   190.4  619.11     200  620.02
   209.5  621.17     219  623.73   228.5  627.37   238.1  631.66   247.6   636.4
   257.1  641.59   266.6  647.21
#Mann= 3 , 0 , 0
       0      .1       0   156.9    .045       0   171.9      .1       0
Bank Sta=156.9,171.9
XS Rating Curve= 0 ,0
Exp/Cntr=0.3,0.1

Type RM Length L Ch R = 1 ,20973   ,123.8,136.8,149.9
XS GIS Cut Line= 2
     1627212.731      510882.092     1627353.567      511107.161
#Sta/Elev= 30
       0  620.93     9.8  620.91    19.7  620.86    29.5  620.48    39.3  618.88
    49.2  615.46    51.4  614.95      59  613.19    66.4  613.31    68.8  613.35
    78.7  614.45    88.5  615.24    98.3  615.59   108.2  615.96     118  616.14
   127.8  616.95   137.7     618   147.5  619.52   157.3  621.34   167.2  623.58
     177  626.31   186.8  629.44   196.7  632.93   206.5  636.55   216.3  640.16
   226.2  643.68     236  647.17   245.8  650.56   255.7  653.99   265.5  657.27
#Mann= 3 , 0 , 0
       0     .06       0    51.4    .045       0    68.8      .1       0
#XS Ineff= 2 , 0
                          109.86             621
Permanent Ineff=
       F       F
Bank Sta=51.4,68.8
XS Rating Curve= 0 ,0
Exp/Cntr=0.3,0.1

Type RM Length L Ch R = 1 ,20836.2 ,180.6,179.8,178.7
XS GIS Cut Line= 2
     1627117.245      510889.036     1627113.984      511161.848
#Sta/Elev= 26
       0  620.64     9.7  620.68    19.5  620.57    29.2  620.27      39  619.74
    48.7  619.02    58.5  617.94    68.2  616.21    78.4  614.11    87.7  613.06
    97.4  613.96   116.9  619.04   126.7  620.67   136.4  622.12   146.2  623.99
   155.9  625.51   165.6  625.85   175.4  625.99   185.1  627.78   194.9  631.04
   204.6  634.16   214.4  636.27   233.9     639   243.6  640.58   263.1  644.08
   272.8  645.72
#Mann= 3 , 0 , 0
       0     .06       0    78.4    .045       0    97.4     .06       0
Bank Sta=78.4,97.4
XS Rating Curve= 0 ,0
Exp/Cntr=0.3,0.1

Type RM Length L Ch R = 1 ,20656.4 ,272.3,248.5,236.8
XS GIS Cut Line= 3
     1626932.349      510733.133     1626940.162      511027.404
     1626971.412      511131.571
#Sta/Elev= 20
       0  620.91     9.8  619.64    19.6  619.02    68.7  617.07   117.8  615.55
   196.2  613.49   240.1  612.14   245.3  612.02   255.1  612.37   264.9  614.03
   274.8  616.69   284.6  619.15   294.4  620.84   303.4  622.53   312.5  625.44
   321.6  629.76   348.8  644.25   375.9  658.82     385  663.64   403.1  673.01
#Mann= 3 , 0 , 0
       0     .06       0   240.1    .045       0   255.1      .1       0
Bank Sta=240.1,255.1
XS Rating Curve= 0 ,0
Exp/Cntr=0.3,0.1

Type RM Length L Ch R = 1 ,20407.9 ,514.2,510.1,493
XS GIS Cut Line= 4
     1626588.599      510714.904      1626664.12      510785.217
      1626757.87      511102.925     1626828.182      511194.071
#Sta/Elev= 30
       0  667.07    18.8  657.64    37.5  648.54    56.3   639.7    84.4  626.84
    93.8  622.98   103.2  619.55   112.9  615.81   122.7  613.64   132.4     613
   142.2   612.9   171.4  612.74   278.6  612.58   307.8  612.18   327.3   611.6
     337  611.48   366.2  611.64   385.7  611.33   395.5  611.44   402.7  612.51
   405.2  612.88     415  615.86   424.7  619.24   434.4  622.01     444  623.85
   453.6  625.44   463.2  628.62   520.8  654.26     540  663.13   549.6  667.73
#Mann= 3 , 0 , 0
       0     .06       0   385.7    .045       0   402.7      .1       0
Bank Sta=385.7,402.7
XS Rating Curve= 0 ,0
Exp/Cntr=0.3,0.1

Type RM Length L Ch R = 1 ,19897.8 ,237.9,249.5,260.7
XS GIS Cut Line= 2
     1626294.328      511030.008     1626505.266       511243.55
#Sta/Elev= 14
       0  650.89    48.4  629.95    58.1  625.65    67.8  620.95    77.5  615.56
    87.1  610.88    93.9  609.53    96.8  608.96   106.5  608.99   108.9  609.13
   116.2  609.54   174.3  613.77   261.4  620.68   300.2  624.03
#Mann= 3 , 0 , 0
       0      .1       0    93.9    .045       0   108.9     .06       0
Bank Sta=93.9,108.9
XS Rating Curve= 0 ,0
Exp/Cntr=0.3,0.1

Type RM Length L Ch R = 1 ,19648.3 ,290.8,291.2,291.4
XS GIS Cut Line= 2
     1626117.245      511110.737      1626226.62       511493.55
#Sta/Elev= 19
       0  650.54    58.3  623.32      68  618.49    77.7  613.15    87.4  608.82
      90  608.32    97.1  606.97   106.8  606.87   116.5  607.28   145.7  608.65
   223.3  612.05   291.3  615.22   330.2  617.34   339.9  618.23   349.6  620.29
     369  627.25   378.7  629.46   388.4  632.37   398.1  637.54
#Mann= 3 , 0 , 0
       0      .1       0      90    .045       0   116.5     .06       0
Bank Sta=90,116.5
XS Rating Curve= 0 ,0
Exp/Cntr=0.3,0.1

Type RM Length L Ch R = 1 ,19357   ,205.3,208.8,212
XS GIS Cut Line= 2
      1625851.62      511222.717     1625944.713      511565.494
#Sta/Elev= 23
       0  649.01      48  623.93    57.6  618.55    67.2  612.38    76.8  607.36
    85.8  605.67    86.4  605.56      96  605.72   100.8  606.06   124.8  608.06
     144     610   172.8  613.22   182.4  614.09     192  614.79   211.2  616.06
   220.8   616.6   230.4  616.96   249.6  617.32   259.2  617.79   278.4  619.04
   307.2  620.67   345.6  623.17   355.2  624.43
#Mann= 3 , 0 , 0
       0      .1       0    85.8    .045       0   100.8     .06       0
Bank Sta=85.8,100.8
XS Rating Curve= 0 ,0
Exp/Cntr=0.3,0.1

Type RM Length L Ch R = 1 ,19148.3 ,265.3,266.6,267.8
XS GIS Cut Line= 2
     1625661.516      511248.758     1625697.974      511558.654
#Sta/Elev= 20
       0  658.41    19.5  647.68    29.2  642.42    68.3   621.8      78  615.95
    87.8  609.89    97.5  606.23   107.3  605.71     117  607.15   121.4  608.21
   136.5   611.9   146.3  613.88     156  615.25   165.8  616.06   175.5  616.45
   204.8  617.08     234  617.86   263.3  618.26     273  618.58     312  620.18
#Mann= 3 , 0 , 0
       0      .1       0    97.5    .045       0   121.4     .06       0
Bank Sta=97.5,121.4
XS Rating Curve= 0 ,0
Exp/Cntr=0.3,0.1

Type RM Length L Ch R = 1 ,18881.7 ,171.8,171.8,171.7
XS GIS Cut Line= 2
     1625404.033      511283.855     1625419.328      511527.404
#Sta/Elev= 28
       0  652.69     9.8  647.24    19.5  641.87    29.3   636.6      39  631.47
    48.8  626.46    58.6   621.4    68.3  615.83    78.1  610.16      87  606.71
    87.8   606.4    97.6  605.68     102  606.15   107.4  606.72   117.1  607.98
   126.9  608.96   136.7  609.71   146.4  610.41   156.2  611.04   165.9  611.58
   175.7  611.97   185.5  612.23   195.2  612.44     205   612.7   214.8  613.04
   224.5   613.4   234.3  613.66     244  613.82
#Mann= 3 , 0 , 0
       0      .1       0      87    .045       0     102     .06       0
Bank Sta=87,102
XS Rating Curve= 0 ,0
Exp/Cntr=0.3,0.1

Type RM Length L Ch R = 1 ,18709.9 ,315.6,293.2,270.5
XS GIS Cut Line= 3
     1625270.234      510992.578     1625233.775      511307.682
       1625249.4      511544.661
#Sta/Elev= 30
       0  703.48     9.6  702.15    38.4  697.63    57.7  694.32    86.5  689.06
   144.2  678.08   153.8  675.98     173  671.22   192.2   666.1   221.1  658.71
   230.7  655.79   240.3     652   249.9  647.39   269.1  637.42   278.8  633.07
   288.4  629.33     298  626.07   317.2  620.22   326.7  617.83   374.2  606.82
   377.5  606.23   383.7  605.13   393.2  604.58   402.7  605.05   431.2  608.59
   440.7   609.3   450.2  609.72   469.2  610.06   497.7  609.95   554.7  610.28
#Mann= 3 , 0 , 0
       0      .1       0   377.5    .045       0   402.7     .06       0
Bank Sta=377.5,402.7
XS Rating Curve= 0 ,0
Exp/Cntr=0.3,0.1

Type RM Length L Ch R = 1 ,18416.7 ,494.7,502.9,505.4
XS GIS Cut Line= 3
     1624729.224      511324.279     1625147.801      511544.071
     1625278.703      511740.946
#Sta/Elev= 30
       0   714.1    48.2  691.25    67.5  682.38    96.5  669.55   125.4  656.55
   173.7  635.92   212.3  619.17   221.9  615.64   231.6  613.54   241.2  612.22
   250.9  610.13   260.5  606.93   270.7  603.81   279.8  602.25   289.4  602.01
   299.1  602.28     328  603.46   424.5   608.2   472.8  610.01   510.6  610.51
   548.4  610.62   576.8  611.15   614.6  612.26   633.5  613.09     643  614.23
   652.4  616.13   661.9  618.76   671.4   621.8   690.3  628.25   709.2  635.49
#Mann= 3 , 0 , 0
       0      .1       0   270.7    .045       0   299.1     .08       0
Bank Sta=270.7,299.1
XS Rating Curve= 0 ,0
Exp/Cntr=0.3,0.1

Type RM Length L Ch R = 1 ,17913.8 ,199.6,204.3,206.8
XS GIS Cut Line= 3
     1624631.307        511687.3     1624856.134       511843.55
     1624928.182      511938.168
#Sta/Elev= 30
       0  621.09     9.8  618.26    19.6  616.55    29.3  615.97    39.1   615.8
    48.9  615.24    58.7  614.32    68.4  613.27      88  610.75    97.8  609.24
   107.6  607.58   117.3  605.72   127.1  603.73   136.9  601.17   144.6  599.67
   146.7  599.26   156.4  598.51   166.2  598.71     176   599.6   185.8  600.81
   234.7  605.86     264  609.04   292.1  611.66   301.2  613.78   310.4  616.79
     347  630.09   365.3  636.95   374.4  640.62   383.6  644.58   392.7  648.79
#Mann= 3 , 0 , 0
       0      .1       0   144.6    .045       0   166.2      .1       0
Bank Sta=144.6,166.2
XS Rating Curve= 0 ,0
Exp/Cntr=0.3,0.1

Type RM Length L Ch R = 1 ,17709.5 ,34.5,33.3,33.2
XS GIS Cut Line= 3
     1624557.523      511669.071      1624572.28      511828.793
     1624738.078      511994.592
#Sta/Elev= 30
       0  642.85    37.7  621.08    47.2  615.88    56.6  611.29      66  608.07
    75.5  606.58    84.9  606.18   113.2  605.65   141.5  604.84     151  604.77
   179.9  605.05   189.7  604.88   199.5  604.56   209.2  602.87     219  599.92
   220.4  599.74   228.8  598.67   235.4  600.48   248.3  603.95   258.1  605.13
   287.4  605.66   297.2  606.02     307  606.56   316.7  607.37   326.5  608.39
   355.8  611.76   365.6  612.54   375.3  613.71   385.1   616.6   394.9  620.75
#Mann= 3 , 0 , 0
       0      .1       0   220.4    .045       0   235.4     .06       0
#XS Ineff= 2 , 0
          179.72  605.66
Permanent Ineff=
       F       F
Bank Sta=220.4,235.4
XS Rating Curve= 0 ,0
Exp/Cntr=0.3,0.1

Type RM Length L Ch R = 1 ,17676.1 ,216.7,231.6,244.8
XS GIS Cut Line= 3
     1624532.349      511690.772     1624547.106      511850.494
     1624712.905      512016.293
#Sta/Elev= 30
       0  633.33     9.4  627.65    18.9  622.26    28.3  617.26    37.7  612.84
    47.2  609.29    56.6   606.8      66  605.33    75.5  604.62    84.9  604.28
   113.2  603.92   122.7  603.73   132.1  603.38   141.5  602.74     151  601.71
   160.4  600.35   189.7  602.08   199.5  602.28   209.2  601.17     219  599.43
   228.8  598.79   236.9  600.51   248.3  602.62   277.6  605.43   287.4  606.34
     307  607.89   365.6  612.38   375.3  613.45   385.1  616.16   394.9  620.96
#Mann= 3 , 0 , 0
       0     .08       0     219    .045       0   236.9     .08       0
#XS Ineff= 2 , 0
          193.24  606.42  249.01          606.58
Permanent Ineff=
       F       F
Bank Sta=219,236.9
XS Rating Curve= 0 ,0
Exp/Cntr=0.3,0.1

Type RM Length L Ch R = 1 ,17444.5 ,307.5,293.5,278.7
XS GIS Cut Line= 2
     1624376.533      511546.241     1624491.551      512090.946
#Sta/Elev= 30
       0  718.25    48.8  697.47    58.6  693.52    78.1  686.53    97.7  678.53
   107.4  674.03   117.2  668.47     127  662.09   136.7  656.55   146.5  653.07
   156.3  651.07     166  647.97   175.8  642.28   185.6  635.46   205.1  621.66
   214.9  614.53   224.6  607.08   234.4  600.75   241.7  598.34   244.2  597.52
   253.9  596.92   263.7  597.08   322.3  598.48   351.6   599.3   400.4  600.76
   429.8  601.88   468.8  603.84   507.9  606.24   537.2  608.29   556.7  609.89
#Mann= 3 , 0 , 0
       0      .1       0   241.7    .045       0   263.7     .06       0
Bank Sta=241.7,263.7
XS Rating Curve= 0 ,0
Exp/Cntr=0.3,0.1

Type RM Length L Ch R = 1 ,17151   ,50,50.9,51.9
XS GIS Cut Line= 2
     1623947.317      511682.682     1624411.255      512123.498
#Sta/Elev= 30
       0  616.17     9.7  614.11    19.4  611.93    29.1  609.62    38.8  607.58
    58.2   605.4    67.9  604.53    87.3   603.9   116.4  603.66   145.4  603.28
   184.2  602.62   203.6  602.57     223  603.15   232.7  602.91   252.1  601.38
   261.8  599.43   268.7  597.93   271.5  597.32   281.2  596.88   290.9  598.01
   310.3   603.6     320  603.61   329.7  603.22   339.4  603.19   397.6  604.18
   426.6  604.44   475.1  605.12   562.4  607.25   610.9  608.64     640  609.67
#Mann= 3 , 0 , 0
       0      .1       0   268.7    .045       0   290.9     .06       0
#XS Ineff= 2 , 0
          224.79  605.42
Permanent Ineff=
       F       F
Bank Sta=268.7,290.9
XS Rating Curve= 0 ,0
Exp/Cntr=0.3,0.1

Type RM Length L Ch R = 1 ,17100.1 ,592.5,591.6,589.1
XS GIS Cut Line= 2
      1624007.61      511806.658     1624380.873      512171.241
#Sta/Elev= 28
       0  607.38    19.3  607.37    38.6  607.53      58  607.85    67.6   607.9
    77.3  607.71      87  607.22    96.6  606.49   106.3  605.93     116  605.22
   125.6  603.29   135.3  599.97   137.1  599.42   144.9  597.06   154.6  597.72
   164.3  599.84   173.9   601.7   183.6  602.18   202.9  602.58   231.9  603.04
   251.2  603.49   309.2  604.26   328.5  604.66   347.8  605.19   367.2  605.88
   405.8  607.02   463.8   608.3   521.8     610
#Mann= 3 , 0 , 0
       0      .1       0   137.1    .045       0   154.6     .06       0
Bank Sta=137.1,154.6
XS Rating Curve= 0 ,0
Exp/Cntr=0.3,0.1

Type RM Length L Ch R = 1 ,16508.5 ,462.4,468.7,474.5
XS GIS Cut Line= 2
     1623710.301       512307.96     1624103.096       512622.63
#Sta/Elev= 27
       0  672.26      29   656.9    38.7  651.95    48.4  647.14    58.1  642.44
    77.4  633.41    87.1  629.13    96.8  624.98   116.1   616.9   125.8  613.06
   135.5  609.48   154.9  602.66   164.5  598.28   168.6  596.61   174.2  594.33
   183.9  592.66   193.6  592.55   203.2  593.07   222.6  595.08   251.6  597.76
     271  599.68   309.7  603.66   464.6  620.32   474.3  621.25   483.9  621.98
   493.6  622.89   503.3  625.67
#Mann= 3 , 0 , 0
       0      .1       0   168.6    .045       0   203.2     .06       0
Bank Sta=168.6,203.2
XS Rating Curve= 0 ,0
Exp/Cntr=0.3,0.1

Type RM Length L Ch R = 1 ,16039.8 ,362.6,352.6,341.6
XS GIS Cut Line= 3
     1623460.338      512635.807     1623585.338      512810.286
     1623806.692      512984.765
#Sta/Elev= 30
       0  633.36    19.5   624.6    48.8  612.18    58.5  607.54    68.3  600.64
      78  594.54    87.8  592.41    97.6  592.46   107.3  593.36   126.8  595.62
   146.3  597.56   175.6  599.86   195.1  601.24   214.6  602.25   224.4  602.56
   234.1  602.37   263.2  600.63     273  600.54   311.8  601.39   370.1  603.18
   389.6  604.15     409  605.38   418.7  607.09   428.4  610.14   438.2  613.66
   447.9  615.89   457.6  617.73   467.3  621.12     477  625.48   496.5  634.58
#Mann= 3 , 0 , 0
       0      .1       0      78    .045       0   107.3     .06       0
#XS Ineff= 2 , 0
                          223.24          603.25
Permanent Ineff=
       F       F
Bank Sta=78,107.3
XS Rating Curve= 0 ,0
Exp/Cntr=0.3,0.1

Type RM Length L Ch R = 1 ,15687.2 ,218.3,217.3,216.1
XS GIS Cut Line= 2
     1623115.682      512880.876      1623705.96      513202.057
#Sta/Elev= 30
       0  636.47      39  622.86    48.7  619.76    58.4  617.45    68.2  616.23
   107.1  614.03   116.9  612.72   126.6  610.34   146.1  603.95   155.8  601.18
   165.6  599.35   175.3  598.13     185  596.16   194.8  593.51   203.2  591.96
   214.3   591.2     224  591.39   301.9  595.37   340.9  596.94   370.1  597.42
     409  597.01   477.2  597.92   545.4  600.53   555.1  602.58   564.9  605.77
   584.4  610.62   594.1  615.01   613.6  625.98   623.3  630.92     672  652.89
#Mann= 3 , 0 , 0
       0      .1       0   203.2    .045       0     224     .06       0
Bank Sta=203.2,224
XS Rating Curve= 0 ,0
Exp/Cntr=0.3,0.1

Type RM Length L Ch R = 1 ,15469.9 ,32.8,32.8,32.7
XS GIS Cut Line= 2
     1623128.993      513127.838     1623610.764      513363.515
#Sta/Elev= 30
       0  623.99     9.8  621.22    19.5  618.27      39  611.78    58.5  604.95
    68.3   601.9      78  599.25    87.8  594.81    97.5  591.76   107.3  591.11
     117  592.32   126.8   593.9   136.5  594.22   146.3  594.43   175.5  594.43
   185.3  594.77   204.8  595.17   214.5   595.6   224.3  595.67     234  596.04
   243.8  595.98   282.8   596.6   292.5  596.51   380.3  598.19   419.3   599.3
   438.8  600.44   468.1  601.73   487.6  603.08   516.8   605.5   536.3   607.5
#Mann= 3 , 0 , 0
       0      .1       0    97.5    .045       0     117     .06       0
#XS Ineff= 2 , 0
                          178.31           600.9
Permanent Ineff=
       F       F
Bank Sta=97.5,117
XS Rating Curve= 0 ,0
Exp/Cntr=0.3,0.1

Type RM Length L Ch R = 1 ,15437.2 ,134.5,133.1,131.8
XS GIS Cut Line= 2
     1623112.066      513155.182     1623593.836      513390.859
#Sta/Elev= 30
       0  631.65     9.8  628.82    19.5  625.74      39  618.78    48.8  615.52
    58.5  612.06    68.3   608.4      78  604.39    87.8  599.68    97.2  594.38
    97.5  594.21   107.3  591.18     117  591.85   126.8  594.36   136.5  596.28
   146.3  597.32     156  597.85   165.8  598.09   185.3  598.27     234   599.2
   341.3   600.2   380.3   600.4   399.8  600.68   409.6  601.16   429.1   602.8
   438.8  602.95   458.3  602.24   468.1  602.32   497.3  603.38   536.3  605.21
#Mann= 3 , 0 , 0
       0      .1       0    97.2    .045       0   126.8     .06       0
Bank Sta=97.2,126.8
XS Rating Curve= 0 ,0
Exp/Cntr=0.3,0.1

Type RM Length L Ch R = 1 ,15304.1 ,231.3,236.2,240.1
XS GIS Cut Line= 2
     1623085.338      513294.661     1623353.567       513406.64
#Sta/Elev= 22
       0   621.9    38.8  604.48    48.4  599.88    58.1  594.83    65.5  592.13
    67.8  591.29    77.5   590.2    87.2  590.93   106.6  594.02   116.3  595.04
     126  595.91   135.6  596.56   145.3  597.08     155  597.52   174.4  597.68
   184.1  597.61   203.5  597.12   213.2  597.01   222.8   597.1   232.5  597.36
   242.2   597.8   290.7  600.28
#Mann= 3 , 0 , 0
       0      .1       0    65.5    .045       0    87.2     .06       0
Bank Sta=65.5,87.2
XS Rating Curve= 0 ,0
Exp/Cntr=0.3,0.1

Type RM Length L Ch R = 1 ,15067.8 ,311.9,312.4,312.3
XS GIS Cut Line= 2
     1622954.079      513465.512     1623329.079       513712.04
#Sta/Elev= 22
       0  644.38     9.8  640.16    19.5   635.7    48.8  621.84    58.5  617.34
      78  608.53    87.8  604.21    97.6  599.63   107.3  594.63   117.1  590.39
     123  589.66   126.8  589.19   136.6  589.37     138  589.46   282.9  599.61
     322  602.16     361  605.12   390.2  607.04     400  608.14   409.8  610.36
   429.3  615.86   448.8  621.53
#Mann= 3 , 0 , 0
       0      .1       0     123    .045       0     138      .1       0
Bank Sta=123,138
XS Rating Curve= 0 ,0
Exp/Cntr=0.3,0.1

Type RM Length L Ch R = 1 ,14755.4 ,217.7,217.5,217.3
XS GIS Cut Line= 2
     1622783.941      513722.456     1623136.371      513960.303
#Sta/Elev= 30
       0  622.25    19.3  614.96    38.6  607.96    48.3  604.82    67.6   599.1
    77.3  596.04      87  592.62    96.6   589.7   106.3  588.72     116  589.01
   120.6  589.37   183.6  594.36   202.9  595.42   222.2  596.13   231.9  596.41
   241.6  596.65   251.2  596.78   270.6  596.81   299.6  596.38   318.9  596.32
   328.6  596.18   338.2  595.82   347.9  595.73   357.5  596.85   367.2  600.18
   386.5  609.86   396.2  612.81   405.8  614.77   415.5  618.25   425.2  622.43
#Mann= 3 , 0 , 0
       0      .1       0    96.6    .045       0   120.6     .08       0
Bank Sta=96.6,120.6
XS Rating Curve= 0 ,0
Exp/Cntr=0.3,0.1

Type RM Length L Ch R = 1 ,14537.9 ,232.5,230,226.9
XS GIS Cut Line= 2
     1622643.316      513887.387     1622999.218      514128.706
#Sta/Elev= 28
       0  626.09    19.6  618.48    29.3   614.8    58.6   603.9    68.4  600.36
    78.2  596.62      88  592.41    97.7  589.26   107.5   588.2   117.3   588.2
   125.7  588.44   156.4  590.03   205.2  592.23   234.6  593.73   263.9   595.5
   283.4  596.86     303  598.39   322.5   600.1   332.3  601.11     342  602.34
   351.8  603.78   361.6  605.42   371.4  607.26   390.9  611.18   400.7  612.99
   410.5  614.23   420.2  614.82     430  615.84
#Mann= 3 , 0 , 0
       0      .1       0   107.5    .045       0   125.7      .1       0
Bank Sta=107.5,125.7
XS Rating Curve= 0 ,0
Exp/Cntr=0.3,0.1

Type RM Length L Ch R = 1 ,14307.9 ,289.1,291.8,294.1
XS GIS Cut Line= 2
     1622515.025      514083.723     1622793.671      514221.744
#Sta/Elev= 20
       0  601.94     9.7  601.51    29.2  600.48    38.9  599.91    58.3  598.61
    87.5  597.02    97.2  596.37   106.9  595.37   116.6   593.1   126.3  589.75
     136  588.74   145.8  591.52   155.5  593.68   165.2  594.31   174.9  594.66
   194.4  594.92   213.8  595.06   252.6  595.11   281.8  595.49     311  595.45
#Mann= 3 , 0 , 0
       0      .1       0   126.3    .045       0   145.8      .1       0
Bank Sta=126.3,145.8
XS Rating Curve= 0 ,0
Exp/Cntr=0.3,0.1

Type RM Length L Ch R = 1 ,14016.2 ,265.2,268.2,270.4
XS GIS Cut Line= 2
     1622257.899      514245.026     1622999.653      514678.994
#Sta/Elev= 30
       0  635.84    29.3  621.89    39.1  617.79    58.6  612.64    68.4  608.93
    87.9  599.15    97.7  595.01   107.4  592.92   136.7  591.49   214.8  589.52
   249.9  587.49   253.9  587.37   264.9  587.45   302.7   588.6     332  590.18
   371.1  592.98   390.6  595.12   410.2  598.79   478.5  616.22     498  619.46
   507.8  622.97   527.3  630.99   615.2  662.02   664.1  680.62   693.4  692.95
   712.9  699.28   732.4  704.51     791  716.98   830.1  724.46   859.4  730.63
#Mann= 3 , 0 , 0
       0      .1       0   249.9    .045       0   264.9      .1       0
Bank Sta=249.9,264.9
XS Rating Curve= 0 ,0
Exp/Cntr=0.3,0.1

Type RM Length L Ch R = 1 ,13747.9 ,130.5,135.8,140.5
XS GIS Cut Line= 2
     1622202.199      514470.648     1622786.111      514849.133
#Sta/Elev= 30
       0  620.48    19.6  611.06    29.4  607.69    39.2  605.81      49  601.96
    58.8  595.48    68.6  590.03    78.4  587.66    88.2  587.35   107.8  587.77
     147  589.76   205.8  592.02     245  593.42   274.4  594.04   313.6  594.51
   362.6  594.31   382.2  593.98   421.4  592.58   431.2  592.59     441  592.91
   460.6  594.96   480.2  594.06     490   594.1   499.8  594.72     539   601.5
   578.2  607.33   617.4  617.55     637  621.28   656.6  623.47   695.8  626.49
#Mann= 3 , 0 , 0
       0      .1       0    68.6    .045       0   107.8      .1       0
Bank Sta=68.6,107.8
XS Rating Curve= 0 ,0
Exp/Cntr=0.3,0.1

Type RM Length L Ch R = 1 ,13612.2 ,30.6,30.1,29.3
XS GIS Cut Line= 4
     1622109.968      514448.512     1622185.923      514605.847
     1622260.792      514683.972     1622481.062      514854.328
#Sta/Elev= 30
       0   662.4    19.4  656.11    29.1  652.81    38.8  649.23    48.5  644.88
    58.2  640.17    67.9  635.23   106.8  614.95   116.5  610.18   126.2  606.55
   145.6  602.36   174.7  593.96   184.6  590.76   192.8  588.64   194.4  588.23
   204.2  587.01   214.1  587.07   263.2  589.29   321.3  591.62   378.9  593.42
   388.5  593.88   417.4  595.64   436.6  596.54   446.2   596.9   465.4   597.3
   494.2  597.41   513.4  597.67   532.6  598.36   542.2  598.88   561.4  600.25
#Mann= 3 , 0 , 0
       0      .1       0   192.8    .045       0   214.1     .06       0
Bank Sta=192.8,214.1
XS Rating Curve= 0 ,0
Exp/Cntr=0.3,0.1

Type RM Length L Ch R = 1 ,13582.1 ,240.5,232.1,223.6
XS GIS Cut Line= 4
     1621965.654      514591.741     1622160.966      514624.294
     1622247.772      514710.014     1622469.126      514874.945
#Sta/Elev= 30
       0  640.81     9.4  636.96    28.3  629.51    37.7  625.98    47.1  622.68
    75.4  613.24    94.3  607.12   103.7  604.33   113.2  602.07   122.6  600.47
     132  599.26   141.4  598.23   150.9  597.27   169.7  595.92     198  593.18
   207.4  591.21   216.8  588.97   221.5  588.12   226.2  587.26   235.5  586.78
   244.9   586.9   358.1   591.9   405.7  593.18   434.2   594.4   481.8   596.2
   510.4  596.94   538.9  597.16     558  597.74     577  598.78     596  600.37
#Mann= 3 , 0 , 0
       0      .1       0   221.5    .045       0   244.9     .06       0
Bank Sta=221.5,244.9
XS Rating Curve= 0 ,0
Exp/Cntr=0.3,0.1

Type RM Length L Ch R = 1 ,13350   ,177.2,179,179.9
XS GIS Cut Line= 2
     1621937.442      514770.778     1622448.509      514986.707
#Sta/Elev= 30
       0  622.28     9.7  616.17    19.5  611.09    29.2  606.74    58.4  597.63
    68.1   594.1    77.9   590.8    87.6   588.7    96.6  587.12   107.1  585.97
   116.8  585.84   155.7  585.81   175.2  586.06   204.4  586.88   272.5  589.95
     292  590.68   360.1  592.06   408.8  593.19   428.3  593.89     438  594.71
   447.7  595.89   457.5  597.31   486.7  602.02   496.4  603.46   506.1  604.72
   515.9  605.71   525.6  606.46   535.3     607   545.1  607.71   554.8  609.75
#Mann= 3 , 0 , 0
       0      .1       0    96.6    .045       0   116.8     .06       0
Bank Sta=96.6,116.8
XS Rating Curve= 0 ,0
Exp/Cntr=0.3,0.1

Type RM Length L Ch R = 1 ,13171   ,124.7,125.9,127.3
XS GIS Cut Line= 2
     1621851.721       514918.13     1622239.742      515103.026
#Sta/Elev= 28
       0  635.81    19.5  626.56    29.3  622.09    48.8   613.6    68.4  605.47
    78.2  601.58    87.9  597.96    97.7  594.41   107.5  591.43   117.2  589.77
     127  588.27   136.8  586.55   146.5  585.59   156.3  585.48   166.1  585.66
   185.6  586.32   205.1  587.21   234.4   588.7   283.3  591.38   312.6  592.86
   332.1  593.68   361.4  594.58   371.2  594.72     381  594.66   390.8   594.2
   410.3  593.63     420  593.78   429.8  594.35
#Mann= 3 , 0 , 0
       0      .1       0   136.8    .045       0   166.1     .06       0
Bank Sta=136.8,166.1
XS Rating Curve= 0 ,0
Exp/Cntr=0.3,0.1

Type RM Length L Ch R = 1 ,13045.1 ,593,586.7,575.6
XS GIS Cut Line= 3
     1620437.659      514532.714     1621739.742       514980.63
     1622192.867      515235.839
#Sta/Elev= 30
       0  862.83      59  845.42   108.2  825.36   157.4  810.92   186.9  806.21
     236  802.52   324.6  801.22   354.1  798.64   383.6   792.4   442.6  774.47
   531.1  752.43   580.3  742.52   629.5  735.61   688.5  714.24   806.5  662.04
     836  650.71   855.7  651.12  1062.2  689.07  1140.9  699.05  1190.1  694.17
  1288.4  697.02  1327.8   682.6    1534  595.61  1553.6   589.8  1577.6  586.49
  1592.6  585.21  1779.3  588.46  1818.5  593.12  1867.6  606.59    1897  611.51
#Mann= 3 , 0 , 0
       0      .1       0  1577.6    .045       0  1592.6     .06       0
Bank Sta=1577.6,1592.6
XS Rating Curve= 0 ,0
Exp/Cntr=0.3,0.1

Type RM Length L Ch R = 1 ,12458.4 ,257.7,254.9,253.5
XS GIS Cut Line= 3
     1620198.075       515449.38     1621505.367      515517.089
     1622036.617      515621.255
#Sta/Elev= 30
       0  661.62    68.9  648.44    98.4  645.77   265.8  649.48   344.5  654.03
   442.9  655.63   511.8  659.19     561   658.1   669.3  652.76     876  651.45
   895.7  650.13   915.4  646.98   974.4  629.11  1053.1  609.69  1072.8  609.27
  1102.4  612.96  1171.2  610.44    1367  594.15  1531.4  588.42  1561.4  581.78
  1570.1  581.26  1579.7  582.11  1599.1  585.48  1676.4  584.94  1724.7  588.13
  1734.4  590.58  1753.7  598.25  1782.7  604.23  1811.7  615.22  1850.4  632.01
#Mann= 3 , 0 , 0
       0     .06       0  1561.4    .045       0  1579.7     .06       0
Bank Sta=1561.4,1579.7
XS Rating Curve= 0 ,0
Exp/Cntr=0.3,0.1

Type RM Length L Ch R = 1 ,12203.4 ,765.2,744.9,722.2
XS GIS Cut Line= 3
     1620807.016      516591.307     1621349.551      515792.696
     1621994.082      515810.057
#Sta/Elev= 30
       0  710.89    58.5  718.35     195  744.57   292.6  757.86   341.3  760.99
   380.3  760.64   409.6  758.27   448.6   753.8   507.1  744.25   575.4  730.99
   633.9  718.11   672.9  711.16   848.4  701.99   887.4  697.91   926.5     691
  1004.5  670.76  1072.9  649.72  1102.2  636.19  1160.8  604.64  1190.2   594.3
  1209.7  590.55    1239  588.31  1317.2  588.99  1348.8  582.23  1356.2  581.57
  1363.8  582.22  1405.1     590  1483.2   597.4  1522.3  610.18  1610.2  643.73
#Mann= 3 , 0 , 0
       0     .06       0  1348.8    .045       0  1363.8     .06       0
Bank Sta=1348.8,1363.8
XS Rating Curve= 0 ,0
Exp/Cntr=0.3,0.1

Type RM Length L Ch R = 1 ,11458.5 ,235.1,244.5,254
XS GIS Cut Line= 3
     1621653.371      516662.922     1621985.402      516270.127
     1622135.141      516205.023
#Sta/Elev= 30
       0  685.88     9.7  686.61    19.4  686.56    48.5  684.35    58.2   683.4
    67.9  681.69    77.6  678.47   106.8  664.33   174.7  626.87   203.8  611.52
   232.9  596.85   242.6  592.44     262  585.13   271.7  580.77   275.1  580.34
   281.4  579.55   290.1  580.49   310.5  584.56   407.6   587.4     427  589.55
   494.9  599.04   523.9  602.45   533.5  605.15   552.8  614.24   562.4  618.17
   581.6  622.25     620   636.3   639.2  640.95   648.8  644.45   677.6  661.13
#Mann= 3 , 0 , 0
       0      .1       0   275.1    .045       0   290.1     .06       0
Bank Sta=275.1,290.1
XS Rating Curve= 0 ,0
Exp/Cntr=0.3,0.1

Type RM Length L Ch R = 1 ,11214   ,399.2,407.5,415
XS GIS Cut Line= 2
     1621874.725       516636.88     1622241.478      516461.099
#Sta/Elev= 30
       0  622.39     9.7  618.44    19.4  614.22      29  609.58    38.7  603.72
    48.4   597.2    58.1  591.89    67.8  589.71    87.2  588.55   125.9  585.62
   145.2  583.99   154.9  582.42   164.6  580.09   174.3  578.58     184  579.38
   186.3  580.08   193.7  582.34   203.4  585.47     213  586.56   222.7  587.26
   232.4  588.58   242.1  590.38   251.8  592.34   280.8  598.78   300.2   603.4
   338.9  612.86   358.3  617.31   377.6  621.42     397  625.02   406.7  626.55
#Mann= 3 , 0 , 0
       0     .08       0   164.6    .045       0   186.3     .06       0
Bank Sta=164.6,186.3
XS Rating Curve= 0 ,0
Exp/Cntr=0.3,0.1

Type RM Length L Ch R = 1 ,10806.5 ,691.1,677,663.4
XS GIS Cut Line= 2
     1621840.003      516984.103     1622308.753       516936.36
#Sta/Elev= 30
       0  630.38    19.6  622.18    49.1  608.59    78.5  595.68    98.2  587.88
     108  585.26   117.8  584.03   127.6  583.66   166.9   583.4     216  583.62
   225.8  583.92   245.4  585.36   255.2  584.46   272.2  578.83   274.8     578
   284.7  577.57   287.2  578.06   304.3  581.59   314.1  582.38   333.8  582.56
   343.6  583.18     373  587.07   382.8  588.53   392.6  590.42   402.5     593
   412.3  596.27   422.1  599.99   441.7  608.01   461.4  616.81   471.2  620.79
#Mann= 3 , 0 , 0
       0     .08       0   272.2    .045       0   287.2     .08       0
Bank Sta=272.2,287.2
XS Rating Curve= 0 ,0
Exp/Cntr=0.3,0.1

Type RM Length L Ch R = 1 ,10129.5 ,362.3,373.6,382.2
XS GIS Cut Line= 3
      1622115.61      517624.294      1622419.43      517398.599
     1622540.957      517329.155
#Sta/Elev= 30
       0  637.01    29.1  622.36    58.2  607.48    67.9  603.02    77.6  599.39
    87.3  595.96      97  591.83   106.8  585.72   116.4     580   126.2  576.72
   135.9  577.26     143  578.94   145.6  579.55   155.3  581.02     165  581.59
   194.1  581.78     262  581.97   291.1   582.9   349.4  585.55   359.1  586.22
   368.8  588.08   378.5   591.1   387.8  594.44   397.1  598.52   406.5  603.19
   415.8  607.96   443.8  621.34   462.5  630.61   471.8  635.04   518.4     655
#Mann= 3 , 0 , 0
       0      .1       0   116.4    .045       0     143     .06       0
Bank Sta=116.4,143
XS Rating Curve= 0 ,0
Exp/Cntr=0.3,0.1

Type RM Length L Ch R = 1 ,9755.8  ,825.4,821.3,814.4
XS GIS Cut Line= 3
     1622191.565       517873.86     1622655.975      517743.651
     1622807.884      517650.335
#Sta/Elev= 30
       0  634.71    19.3  629.13    38.6  622.17   106.1  593.89   115.8  590.93
   125.4  588.77     135  587.33   154.3  585.87   173.6  585.74   202.6  586.45
   221.9  586.05   270.1  582.24   299.3  576.33   308.7  575.78   314.3  575.81
     328  576.36   376.2  580.16   385.8  582.28   405.2  588.68   414.8  590.23
   424.4  589.79   443.7  584.74   453.4  584.85     463  587.64   472.7  591.43
   482.3  595.85   538.6  626.66   594.9  655.22   632.4  673.02   660.6  684.17
#Mann= 3 , 0 , 0
       0      .1       0   299.3    .045       0   314.3      .1       0
Bank Sta=299.3,314.3
XS Rating Curve= 0 ,0
Exp/Cntr=0.3,0.1

Type RM Length L Ch R = 1 ,8934.5  ,1226.7,1230.1,1233.9
XS GIS Cut Line= 2
     1622418.272      518604.762     1622987.717      518375.596
#Sta/Elev= 30
       0  670.36    48.7  649.12    87.7  632.77   116.9  620.86   165.6  601.72
   175.4  598.07   185.1  594.76   224.1  583.01   233.8  580.43   243.6  579.05
   253.3   578.8   292.3  578.95   350.8  579.84   360.5  579.83   370.2  578.86
     380  576.38   389.7  573.59   399.5  572.46   407.8  572.81   422.8  574.23
   457.9     578   467.7  579.48   477.4  582.55   487.2  587.52   526.1  611.72
   535.9  617.56   545.6  623.08   555.4  628.18   565.1  632.91   613.8  655.38
#Mann= 3 , 0 , 0
       0      .1       0   407.8    .045       0   422.8      .1       0
Bank Sta=407.8,422.8
XS Rating Curve= 0 ,0
Exp/Cntr=0.3,0.1

Type RM Length L Ch R = 1 ,7704.4  ,748.3,738.6,726.6
XS GIS Cut Line= 2
     1622810.633      519576.985     1623293.272      519392.957
#Sta/Elev= 30
       0  669.33    48.7  644.62      78   630.6    87.7  626.22   126.7  609.91
   146.2  601.39   155.9  597.32   165.7  593.53   175.4  590.16   185.2  587.21
   194.9   584.6   204.7  582.38   214.4   580.6   224.2  579.11   233.9  578.04
   253.4  576.76   263.1  574.76   272.9  572.14   282.6  570.03   284.2  569.99
   292.4  569.79   299.2  570.13   311.9  571.34   331.4  574.32   380.1  579.19
   389.8  580.53   409.3  584.51   438.6  591.22   487.3  601.65   516.5  608.23
#Mann= 3 , 0 , 0
       0      .1       0   284.2    .045       0   299.2      .1       0
Bank Sta=284.2,299.2
XS Rating Curve= 0 ,0
Exp/Cntr=0.3,0.1

Type RM Length L Ch R = 1 ,6965.8  ,386.6,386,385.2
XS GIS Cut Line= 2
     1623317.578      520229.762     1623730.772      519826.985
#Sta/Elev= 30
       0  644.44     9.8  639.68    19.6   635.3    68.5  615.22   136.9  586.02
   156.5  578.32   166.3  575.58     176  575.11   224.9   575.1   244.5   575.2
   283.6  575.92   293.4  575.24   303.2  572.86   313.2  569.64   322.7  568.41
   332.5  569.12   342.3  571.22   352.1  573.01   361.9   574.4   371.6  575.44
   391.2  576.39   420.5  577.01   430.3  577.65   440.1  579.92   449.9  584.36
   459.7  589.72     489  606.29   537.9  633.52   567.2  650.72     577  656.12
#Mann= 3 , 0 , 0
       0      .1       0   313.2    .045       0   332.5      .1       0
Bank Sta=313.2,332.5
XS Rating Curve= 0 ,0
Exp/Cntr=0.3,0.1

Type RM Length L Ch R = 1 ,6579.8  ,619.6,623.4,624.9
XS GIS Cut Line= 2
     1623577.994       520507.54     1623956.467       520101.29
#Sta/Elev= 30
       0  588.01    58.4  589.07    77.9  589.19   146.1  588.59   155.8  587.99
   165.6  586.24   175.3   583.8   185.1  582.06   194.8  581.76   233.8   581.7
   243.5  581.57   253.3  580.88     263  577.08   272.7  571.39   281.2  567.86
   282.5  567.32   292.2  567.55   296.2  568.36   311.7  571.34   321.4   572.1
   350.7  573.42   409.1  575.77   428.6  576.65   457.8  578.28     487   580.2
   496.8  581.02     526  584.57   535.8  585.62   545.5  586.86   555.2  587.79
#Mann= 3 , 0 , 0
       0      .1       0   281.2    .045       0   296.2      .1       0
Bank Sta=281.2,296.2
XS Rating Curve= 0 ,0
Exp/Cntr=0.3,0.1

Type RM Length L Ch R = 1 ,5956.4  ,5917.4,5956.4,5985.4
XS GIS Cut Line= 2
     1623935.633      520906.846     1624373.133      520531.846
#Sta/Elev= 30
       0  581.47    19.5  581.56    48.8  581.25   136.7  579.72     166  579.61
   175.8  579.78   185.6  579.62   195.3  578.08   214.9  573.26   224.6  572.18
   234.4  571.92   273.5   571.7     293  571.25   312.5  570.17   322.3  569.37
   351.6  566.38   360.6  566.14   361.4  566.12   371.1  566.22   375.6  566.71
   380.9  567.28   390.7  571.59     420  588.84   449.3  606.74   468.8  619.04
   498.1   638.2   517.6  650.47   537.2  661.72   546.9  667.03   576.2  682.48
#Mann= 3 , 0 , 0
       0     .08       0   360.6    .045       0   375.6      .1       0
Bank Sta=360.6,375.6
XS Rating Curve= 0 ,0
Exp/Cntr=0.3,0.1

Chan Stop Cuts=-1
Use User Specified Reach Order=0
Composite Channel Slope=5
